--- GRFTHCK.prj (project) ---

Proj Title=GRFTHCK
Current Plan=p01
Default Exp/Contr=0,0
English Units
Geom File=g01
Flow File=f01
Plan File=p01
BEGIN DESCRIPTION:
END DESCRIPTION:
DSS Export Rating Curves= 0
DSS Export Rating Curve Sorted= 0
DSS Export Volume Flow Curves= 0
DXF OffsetX= 0
DXF OffsetY= 0
DXF ScaleX= 0
DXF ScaleY= 0

--- GRFTHCK.p01 (plan) ---

Plan Title=Floodplain
Program Version=4.00
Geom File=g01
Flow File=f01
K Sum by GR=0
Std Step Tol=0.01
Critical Tol=0.01
Num of Std Step Trials=20
Max Error Tol=0.3
Flow Tol Ratio=0.001
Split Flow NTrial=30
Split Flow Tol=0.02
Split Flow Ratio=0.02
Log Output Level=0
Friction Slope Method=1
Unsteady Friction Slope Method=2
Unsteady Bridges Friction Slope Method=1
Global Log Level=0
CheckData=False
Run HTab=0
Run UNet=0
Run PostProcess=0
UNET Theta=0
UNET Theta Warmup=0
UNET ZTol=0
UNET ZSATol=0
UNET MxIter=0
UNET MaxInSteps=0
UNET DtIC=0
UNET DtMin=0
UNET MaxCRTS=0
UNET WFStab=0
UNET SFStab=0
UNET WFX=0
UNET SFX=0
UNET DSS MLevel=0
UNET DZMax Abort=0
UNET Convert EG Bridges=0
UNET Use Existing IB Tables=0
UNET Froude Limit=0
UNET Froude Power=0
Write IC File=0
Echo Input=False
Echo Output=False
Write Detailed=0

--- GRFTHCK.f01 (steady flow) ---

Flow Title=2010 USGS WV Regression Equation
Program Version=4.10
Number of Profiles= 1
Profile Names=P100yr
River Rch & RM=GRFTHCK,Main            ,10392.9
379.0315
River Rch & RM=GRFTHCK,Main            ,9726.8
403.1947
River Rch & RM=GRFTHCK,Main            ,7346.6
429.8254
River Rch & RM=GRFTHCK,Main            ,4912.6
476.5972
River Rch & RM=GRFTHCK,Main            ,4800.5
628.0701
River Rch & RM=GRFTHCK,Main            ,2195
645.2995
River Rch & RM=GRFTHCK,Main            ,1882.2
724.6715
River Rch & RM=GRFTHCK,Main            ,147.8
789.0615
Boundary for River Rch & Prof#=GRFTHCK,Main            , 1
Up Type= 0
Dn Type= 1
Dn Known WS=1712
DSS Import GetInterval= 0
DSS Import GetPeak= 0
DSS Import FillOption= 0

--- GRFTHCK.g01 (geometry) ---

Geom Title=LiDAR
Program Version=4.10

River Reach=GRFTHCK         ,Main
Reach XY= 30
     2049276.512      273047.418     2049316.402      272796.164
     2049198.781      272640.348      2049115.02      272220.902
     2049307.777       272106.78     2049304.149      271892.758
     2049645.392      271620.459     2049850.471      271220.069
      2050079.42      271116.987     2050145.571      270781.951
     2050492.078      270268.984      2050481.11      270130.108
     2050867.617      270035.747     2050960.933      269892.084
     2051387.149      269744.514     2051647.813      269498.593
     2051788.475      269513.254     2052390.618      269283.003
     2052426.645      269066.997     2052676.643       268895.85
     2053020.393      268331.614     2053353.596      268072.195
     2053620.318      268006.933     2053915.996      267723.119
      2054131.94      267698.941     2054333.531      267480.932
     2054362.654      267233.862     2054526.016      267257.907
     2054736.401       267157.68     2055308.988      266456.202

Type RM Length L Ch R = 1 ,10392.9 ,224.1,230.7,236.6
XS GIS Cut Line= 3
     2049496.519      273035.152     2049302.508      273022.132
     2049065.529      273080.725
#Sta/Elev= 30
       0 2178.56    19.4 2169.35    35.6 2160.33    58.3 2151.31    68.1  2146.5
    90.7 2133.35   129.6 2108.56   145.8 2099.29   155.6 2094.58     162 2092.36
   168.5 2091.37     201 2091.46   220.5  2086.9     227 2086.58   230.2 2086.87
  231.682087.501   233.5 2088.28   246.5 2098.98  271.112101.987   275.8 2103.43
   282.3 2106.76   301.9 2106.18   314.9 2104.75   337.7 2104.72   360.4 2106.74
  379.73 2110.84   402.8 2118.39   412.5 2122.68   429.82131.872   438.6 2136.82
#Mann= 7 ,-1 , 0
       0     .12       0   220.5    .045       0   230.2     .12       0
  231.68    .016       0  271.11     .12       0  379.73     .06       0
   429.8     .12       0
Bank Sta=220.5,230.2
XS Rating Curve= 0 ,0
Exp/Cntr=0.3,0.1

Type RM Length L Ch R = 1 ,10162.1 ,105.9,91,75.7
XS GIS Cut Line= 3
     2049495.216      272819.007     2049233.498      272809.892
     2049021.258       272864.58
#Sta/Elev= 30
       0 2169.75    32.7 2150.94    42.6 2149.42    45.8 2148.08    65.5 2136.59
    88.4 2126.32    98.2 2121.31   121.1 2106.56   134.2  2098.8   147.3 2089.78
   150.6 2088.13   157.1 2086.53   173.5 2076.92   176.8 2076.15  184.262076.919
     216 2085.04   229.1  2089.3   242.2 2090.57  251.91 2090.74   265.2 2090.87
     288 2093.14  308.67 2093.52   373.1 2097.08   392.7 2097.51  408.462099.179
   418.9 2101.67     432 2105.96     4602118.081   474.5 2123.65     481 2125.45
#Mann= 7 ,-1 , 0
       0     .12       0   173.5    .045       0  184.26     .12       0
  251.91    .016       0  308.67     .12       0  408.46     .06       0
     460     .12       0
Bank Sta=173.5,184.26
XS Rating Curve= 0 ,0
Exp/Cntr=0.3,0.1

Type RM Length L Ch R = 1 ,10071.1 ,112.7,121.3,129.2
XS GIS Cut Line= 3
     2049427.477      272626.559     2049223.559      272775.577
     2049015.719      272839.628
#Sta/Elev= 30
       0 2141.35    16.4 2138.35    42.6 2131.34    52.5 2127.82    68.9 2119.96
    95.1  2112.1   111.5 2102.83   134.5 2086.59   144.3 2083.53   150.9 2078.78
   154.2 2077.22     164 2074.71   170.6 2074.11   177.1 2073.97   183.7 2074.11
   200.1 2076.37   213.2 2083.42     223 2086.85  228.052087.769   249.3 2088.37
  261.152089.961  276.992090.454   301.3 2090.72   346.7 2094.18  365.732094.817
   388.9 2096.11   398.82097.409   411.6 2100.74  452.71 2116.24     470  2120.2
#Mann= 9 ,-1 , 0
       0     .12       0   170.6    .045       0   183.7     .12       0
  228.05    .016       0  261.15     .12       0  276.99    .016       0
  365.73     .12       0   398.8     .06       0  452.71     .12       0
Bank Sta=170.6,183.7
XS Rating Curve= 0 ,0
Exp/Cntr=0.3,0.1

Type RM Length L Ch R = 1 ,9949.8  ,225.2,223,219.6
XS GIS Cut Line= 3
       2049422.3      272582.027     2049144.956       272658.85
      2049016.05      272816.402
#Sta/Elev= 30
       0 2137.04    13.1 2132.93    32.7 2132.26    75.2  2117.6    91.6 2112.97
   104.6 2107.97   114.5 2102.97   140.6 2084.78   153.7 2077.44   160.2 2075.69
   170.1 2076.42   176.6 2075.41     193 2067.22   209.3 2065.47   222.42060.787
   228.9 2060.32  236.222060.788     242 2063.03   255.1 2073.12   268.2 2074.94
  275.682082.285   281.2 2084.58  359.382090.738  409.772092.022   436.4 2095.32
   442.9 2097.34  449.512100.674  473.552108.593  481.17 2110.84   491.4 2113.57
#Mann= 9 ,-1 , 0
       0     .12       0   222.4    .045       0  236.22    .016       0
  275.68     .12       0  359.38     .06       0  409.77    .016       0
  449.51     .12       0  473.55     .06       0  481.17     .12       0
Bank Sta=222.4,236.22
XS Rating Curve= 0 ,0
Exp/Cntr=0.3,0.1

Type RM Length L Ch R = 1 ,9726.8  ,262.2,295,327.8
XS GIS Cut Line= 4
     2049396.258      272481.767      2049210.06      272410.152
     2049036.883      272484.371     2048906.675      272499.996
#Sta/Elev= 30
       0 2119.89    13.1  2116.3    19.6 2112.37    22.9  2111.4    42.5 2109.06
    62.1 2101.33    91.6 2091.74   124.3 2082.82   150.4 2077.49   183.1 2064.58
   212.5 2061.85   225.5 2062.36     232 2059.95   238.5 2053.65   241.7 2052.07
   251.5 2051.18     258 2050.65   264.5  2051.2   274.2 2055.66  282.722057.369
   303.4 2056.39   313.2 2060.76  317.762061.514   332.7 2063.25   342.4 2069.12
   348.9 2071.12   397.7 2078.62   417.4 2084.51   446.9 2096.08     519  2130.2
#Mann= 5 ,-1 , 0
       0     .12       0   251.5    .045       0   264.5     .12       0
  282.72    .016       0  317.76     .12       0
Bank Sta=251.5,264.5
XS Rating Curve= 0 ,0
Exp/Cntr=0.3,0.1

Type RM Length L Ch R = 1 ,9431.8  ,220.1,198.7,176.7
XS GIS Cut Line= 4
     2049431.414      272347.652     2049213.966      272251.298
     2049137.144      272117.184      2048953.55      272106.767
#Sta/Elev= 30
       0 2114.03    16.3 2109.58    39.1 2101.65    65.2 2090.49    78.2 2088.04
   107.5  2076.5   123.8 2071.57   143.4 2067.76   218.3 2062.79   237.8  2053.3
   257.2 2045.73   282.9 2043.16   305.5 2043.87  317.022041.648   320.7 2040.88
     328 2040.16  332.932040.868   337.7 2042.84   350.5 2043.72  358.672046.374
   366.6 2048.33   402.1 2049.27   434.3 2052.61   440.8 2054.53   479.5  2080.6
   492.4 2087.63   518.2 2107.35   531.1 2111.09   556.9 2130.29   576.3 2137.73
#Mann= 5 ,-1 , 0
       0     .12       0  317.02    .016       0   320.7    .045       0
  332.93    .016       0  358.67     .12       0
#XS Ineff= 2 , 0
          303.41 2046.59
Permanent Ineff=
       F       F
Bank Sta=320.7,332.93
XS Rating Curve= 0 ,0
Exp/Cntr=0.3,0.1

Type RM Length L Ch R = 1 ,9233.1  ,99.1,74.7,43.9
XS GIS Cut Line= 4
     2049512.022      272205.222     2049357.508      272069.806
     2049272.439      272061.125     2049031.119      271977.792
#Sta/Elev= 30
       0 2102.92    35.9 2088.57    58.7 2081.63    97.8 2072.83   127.2 2068.91
   143.5 2064.38   166.3 2061.15   205.5  2050.8   208.6 2049.59     215 2043.41
   227.6 2034.96   232.7 2034.18   243.5 2033.64   247.7 2034.07     253 2035.78
  268.722036.515   275.1 2037.12     291 2035.03  305.122037.259   356.4 2039.36
   366.2 2042.81   389.2 2045.28   402.2 2051.01   415.4 2053.36   431.7 2065.09
   454.6 2078.77   461.2 2084.28   503.7 2109.96   510.3 2112.83   546.3 2122.06
#Mann= 5 ,-1 , 0
       0     .12       0   232.7    .045       0   247.7     .12       0
  268.72    .016       0  305.12     .12       0
#XS Ineff= 2 , 0
                          255.11         2038.65
Permanent Ineff=
       F       F
Bank Sta=232.7,247.7
XS Rating Curve= 0 ,0
Exp/Cntr=0.3,0.1

Type RM Length L Ch R = 1 ,9158.4  ,48.1,45.4,51.3
XS GIS Cut Line= 4
     2049586.362      271998.694     2049384.638      271903.711
     2049285.581      272045.569     2049042.091      271957.027
#Sta/Elev= 30
       0 2078.65    16.4 2070.98    36.1 2067.56    62.3 2056.46    88.5    2048
   121.3 2043.75   147.6 2035.12   186.9 2030.03  219.582029.125     223 2028.96
     285 2031.17   311.1 2035.87   317.6 2034.91  326.442030.802  339.222030.802
   363.3 2034.71   405.8 2034.49  416.412035.569   464.9 2038.03   474.7  2041.2
   497.7 2045.31   510.8 2050.63   523.9  2053.6   527.2 2055.46     537 2064.05
   573.1 2086.47   582.9 2093.89   612.4 2112.75   635.4 2124.35   655.1 2130.56
#Mann= 5 ,-1 , 0
       0     .12       0  219.58    .016       0  326.44    .045       0
  339.22    .016       0  416.41     .12       0
#XS Ineff= 2 , 0
          313.52 2038.04
Permanent Ineff=
       F       F
Bank Sta=326.44,339.22
XS Rating Curve= 0 ,0
Exp/Cntr=0.3,0.1

Type RM Length L Ch R = 1 ,9113    ,110.8,152.5,190.9
XS GIS Cut Line= 4
     2049560.321      271962.236     2049358.596      271867.252
     2049259.539      272009.111     2049048.602      271932.288
#Sta/Elev= 30
       0 2062.49    36.1 2048.76    78.7 2040.89   108.2 2030.97   127.9  2031.8
   137.7 2028.73  177.06 2028.02   190.2 2026.52   206.6 2026.36  216.01 2026.98
     223 2028.22   265.4 2027.81   304.6 2031.11   324.2  2028.8   337.2 2028.81
   350.3 2031.73   412.3 2034.96     435  2038.2   454.6 2043.62   464.3 2049.19
   474.1 2051.64   483.8 2057.09   490.3 2059.14   493.6 2061.25   503.4 2070.61
   522.9 2081.21   558.7  2102.6   574.9 2113.52   604.2 2129.88   620.5 2136.82
#Mann= 5 ,-1 , 0
       0     .12       0  177.06    .016       0  216.01     .12       0
   324.2    .045       0   337.2     .12       0
#XS Ineff= 2 , 0
          305.57 2032.97
Permanent Ineff=
       F       F
Bank Sta=324.2,337.2
XS Rating Curve= 0 ,0
Exp/Cntr=0.3,0.1

Type RM Length L Ch R = 1 ,8960.4  ,287.9,297.2,305.2
XS GIS Cut Line= 3
     2049561.623      271937.496     2049387.144      271852.861
     2049208.758      271695.309
#Sta/Elev= 30
       0  2054.2    25.9 2045.36      42 2041.79    67.9 2038.19    80.8 2035.25
    93.7 2029.54      97 2028.74   116.4 2028.11     126 2027.04   148.7 2026.99
  159.49 2026.24     181 2024.48   190.7  2024.7  200.952026.428   203.7 2025.72
   210.2 2021.83   213.5 2020.73   216.7 2020.32  226.842020.729   239.6 2025.35
   252.6 2026.66   268.9 2035.97     282 2042.18   337.4  2061.2   360.2 2072.23
   366.7 2076.17     383 2079.86   402.6 2088.09   422.1 2092.39   431.9 2096.45
#Mann= 5 ,-1 , 0
       0     .12       0  159.49    .016       0  200.95     .12       0
   213.5    .045       0  226.84     .12       0
Bank Sta=213.5,226.84
XS Rating Curve= 0 ,0
Exp/Cntr=0.3,0.1

Type RM Length L Ch R = 1 ,8663.2  ,258.4,244.1,229.5
XS GIS Cut Line= 3
     2049669.696      271807.288     2049562.925      271595.048
     2049353.289      271510.413
#Sta/Elev= 30
       0 2041.21      13 2035.55      26 2031.82    58.6 2028.26    91.1 2018.81
   110.7 2018.22  136.672013.367   143.2 2011.49   156.2 2010.86   166.9  2007.4
   175.8 2006.45  179.982007.369   188.8 2010.34   198.5 2011.36   214.8 2010.17
   221.3 2010.45   227.8  2011.6   237.6 2014.86   257.2 2024.23   276.9 2026.54
     290 2028.91     326 2040.62   365.4    2059   375.2 2065.33   378.5 2066.87
   388.3 2069.03   391.6 2070.42   401.4  2077.3   430.9 2091.48   463.7 2108.42
#Mann= 4 ,-1 , 0
       0     .12       0  136.67    .016       0   166.9    .045       0
  179.98     .12       0
Bank Sta=166.9,179.98
XS Rating Curve= 0 ,0
Exp/Cntr=0.3,0.1

Type RM Length L Ch R = 1 ,8419.1  ,230.6,231.8,230.1
XS GIS Cut Line= 2
     2049889.748      271541.663     2049534.279      271361.975
#Sta/Elev= 30
       0 2043.13    22.8 2029.37    45.7  2018.8    55.5    2016    81.6 2012.37
    84.9 2010.91    91.4 2005.18    97.9 2000.94  107.712000.122   114.3 2001.28
   130.6 2001.39  149.142002.984     160  2003.3     173 2002.15  185.68  1997.5
   189.4 1997.31   199.2 1997.46     209 1998.82  221.472004.101   235.1 2005.15
   244.9 2008.43  256.942014.208   267.7 2018.19   293.8 2021.18   329.7 2029.21
   342.8 2030.57   352.6 2034.52   368.9 2038.58   378.7 2042.39   398.3 2042.58
#Mann= 7 ,-1 , 0
       0     .12       0  107.71    .016       0  149.14     .12       0
  185.68    .045       0   199.2     .12       0  221.47    .016       0
  256.94     .12       0
Bank Sta=185.68,199.2
XS Rating Curve= 0 ,0
Exp/Cntr=0.3,0.1

Type RM Length L Ch R = 1 ,8187.3  ,293.6,296.2,299.3
XS GIS Cut Line= 3
     2049961.362      271442.705     2049849.383      271265.621
     2049635.841      271166.663
#Sta/Elev= 30
       0 2034.85    29.5 2017.12    42.6 2011.27    55.6 2008.26    85.1 2003.48
  106.021995.848   117.8 1994.55     131 1994.71  149.021992.797   157.1 1992.61
   170.2 1989.87   189.9 1987.49   209.5 1989.78   225.9 1989.21   235.7 1988.58
   238.9 1989.13   245.5 1993.24   248.7 1994.17   261.8 1994.65  277.36 2000.09
   284.7 2003.08     301 2008.26   333.7  2015.6   363.2 2024.01   379.5 2026.24
   392.6 2030.22   405.6 2035.13   418.7 2042.46   428.5 2045.94   444.9 2054.56
#Mann= 6 ,-1 , 0
       0     .12       0  106.02    .016       0  149.02     .12       0
   225.9    .045       0   238.9    .016       0  277.36     .12       0
#XS Ineff= 2 , 0
          208.98 1991.76
Permanent Ineff=
       F       F
Bank Sta=225.9,238.9
XS Rating Curve= 0 ,0
Exp/Cntr=0.3,0.1

Type RM Length L Ch R = 1 ,7891.1  ,290.4,279.5,268.1
XS GIS Cut Line= 4
     2050184.019      271296.871     2050100.685      271151.038
     2049910.581       271027.34     2049729.591      271016.923
#Sta/Elev= 30
       0 2054.48    67.8 2020.57      84 2014.92  144.051999.489   158.3 1993.38
   177.7  1992.4   180.9  1990.8  186.23 1984.69   190.6 1978.04  196.441973.579
   200.4 1973.13   210.1 1973.55   226.3 1974.89     236 1979.94   258.7 1978.89
   268.4 1983.06   278.1 1984.75   323.5  1982.8   349.4  1978.4  369.79 1978.98
  415.191980.164   430.4 1980.84     453 1990.86     466  1993.4   478.9 1999.31
   501.6 2011.61   540.4 2039.17   559.9 2043.41   569.6 2052.36   576.1 2055.99
#Mann= 7 ,-1 , 0
       0     .12       0  144.05    .016       0  186.23     .12       0
  196.44    .045       0   210.1     .12       0  369.79    .016       0
  415.19     .12       0
Bank Sta=196.44,210.1
XS Rating Curve= 0 ,0
Exp/Cntr=0.3,0.1

Type RM Length L Ch R = 1 ,7611.6  ,254.1,265,275.6
XS GIS Cut Line= 3
     2050340.269      270880.205     2050049.904      270854.163
     2049858.498      270736.975
#Sta/Elev= 30
       0 1972.53    13.1 1973.51    22.9 1975.94   35.711976.128      59 1976.31
    72.1 1973.54    85.2 1967.68    91.7  1966.8   108.1 1968.64     131 1966.93
   150.7 1967.69   167.1 1966.92   176.9  1969.1   180.2 1968.75     190 1961.68
  195.731960.654   199.8 1960.29   209.8 1960.63   255.5 1968.58  275.361968.849
   301.3 1968.58   320.8 1975.27   327.3 1976.51  362.731976.065  384.521975.699
  430.511977.307   437.9 1978.03  459.711992.782   480.2 2006.66     516 2033.99
#Mann= 9 ,-1 , 0
       0    .016       0   35.71     .12       0  195.73    .045       0
   209.8     .12       0  275.36    .016       0  362.73     .12       0
  384.52    .016       0  430.51     .06       0  459.71     .12       0
Bank Sta=195.73,209.8
XS Rating Curve= 0 ,0
Exp/Cntr=0.3,0.1

Type RM Length L Ch R = 1 ,7346.6  ,249.6,246.4,243.3
XS GIS Cut Line= 3
     2050392.352      270720.048     2050098.081      270535.152
     2049919.696      270557.288
#Sta/Elev= 30
       0 1965.69    62.3 1964.83    68.8 1963.12      82 1956.56    88.5 1954.79
   108.2 1953.29   137.7 1954.71   160.6 1954.34   163.9 1953.66   170.5 1949.26
     177 1947.92  184.241949.372   196.7 1955.98   203.3 1957.24  211.891957.233
     223 1956.58  243.411957.511  322.251963.136  346.511965.383  394.611968.374
   403.1  1968.8   412.9  1971.2   429.2 1978.62  460.481996.222   465.2 1998.91
     475 2001.44   478.3 2003.42   484.8 2009.76   488.1 2011.94   527.3  2031.6
#Mann= 9 ,-1 , 0
       0     .12       0   170.5    .045       0  184.24     .12       0
  211.89    .016       0  243.41     .12       0  322.25     .06       0
  346.51    .016       0  394.61     .06       0  460.48     .12       0
Bank Sta=170.5,184.24
XS Rating Curve= 0 ,0
Exp/Cntr=0.3,0.1

Type RM Length L Ch R = 1 ,7100.2  ,361.1,372.8,379.2
XS GIS Cut Line= 3
     2050529.071      270522.132     2050402.769      270428.382
     2050048.602      270269.527
#Sta/Elev= 30
       0 1960.89    2.79 1960.45    22.9 1956.29      59 1951.76    88.5 1949.92
   101.6 1947.16   131.1 1943.82   143.1 1944.18  150.011944.566   176.9 1943.98
   186.6 1941.05   199.7 1940.24  205.111938.458   209.5 1938.02   219.3 1938.48
     229 1943.39  242.521942.754   261.7 1942.87   274.7 1948.88  287.711951.531
   307.3 1951.65  320.211954.189  346.311956.339  377.491957.501   395.4 1957.28
  426.891961.018   444.3 1965.18   457.4 1971.78   525.9 2018.14   545.4 2029.98
#Mann= 12 ,-1 , 0
       0    .016       0    2.79     .12       0   143.1     .06       0
  150.01     .12       0  205.11    .045       0   219.3     .12       0
  242.52    .016       0  287.71     .12       0  320.21    .016       0
  346.31     .12       0  377.49     .06       0  426.89     .12       0
Bank Sta=205.11,219.3
XS Rating Curve= 0 ,0
Exp/Cntr=0.3,0.1

Type RM Length L Ch R = 1 ,6727.4  ,357.7,366.8,376.1
XS GIS Cut Line= 4
     2050626.657      270423.468     2050560.685      270182.149
      2050411.38       270034.58     2050334.991      269862.705
#Sta/Elev= 30
       0 1951.51    17.51948.847    45.5 1941.68   81.45 1940.71     130 1940.32
   159.2 1935.37  182.671934.882  203.571933.925   217.7  1934.7   233.9 1931.43
   246.9 1931.43  266.231929.214   296.1  1928.1  308.021926.015   315.8 1926.22
  324.21 1924.22   332.2 1923.71  337.091924.219   345.3 1924.64   355.1 1930.53
   391.2 1930.23   410.9 1932.82     424 1932.72   433.9 1934.91     486 1938.33
   518.5  1954.9   550.9 1974.82   580.1 1988.61   615.8 2001.14   648.2 2008.58
#Mann= 9 ,-1 , 0
       0     .12       0    17.5    .016       0   81.45     .12       0
  182.67     .06       0  203.57     .12       0  266.23    .016       0
  308.02     .12       0  324.21    .045       0  337.09     .12       0
#XS Ineff= 2 , 0
          315.69 1928.61
Permanent Ineff=
       F       F
Bank Sta=324.21,337.09
XS Rating Curve= 0 ,0
Exp/Cntr=0.3,0.1

Type RM Length L Ch R = 1 ,6360.6  ,197.8,192.4,186.3
XS GIS Cut Line= 4
     2051038.116      270246.385      2050888.81      270124.857
     2050791.588      269906.107     2050633.602      269763.746
#Sta/Elev= 30
       0 1973.78    29.4 1965.13    88.1 1942.14   140.3 1926.84   169.7 1920.72
  216.021919.738   228.6 1920.28   238.4 1918.33  257.711921.404   264.7 1920.77
   274.5 1911.64  275.981911.089   284.3 1910.02   290.9 1910.99   297.4 1912.34
   323.7 1908.92   349.9 1909.85   359.8 1908.98   379.4 1914.18   415.5 1913.65
   425.3 1916.57     445 1917.36   464.6 1924.81   490.8 1931.07     530 1947.17
   575.8 1964.16   598.8 1976.41   608.6 1985.46   615.1 1989.87   644.6 2004.89
#Mann= 5 ,-1 , 0
       0     .12       0  216.02    .016       0  257.71     .12       0
  275.98    .045       0   290.9     .12       0
#XS Ineff= 2 , 0
                          299.07         1915.81
Permanent Ineff=
       F       F
Bank Sta=275.98,290.9
XS Rating Curve= 0 ,0
Exp/Cntr=0.3,0.1

Type RM Length L Ch R = 1 ,6168.2  ,143.8,148.3,151.6
XS GIS Cut Line= 3
     2051137.348      270107.566     2050888.867      269799.406
     2050751.063       269695.24
#Sta/Elev= 30
       0 1971.59    16.4 1966.62    65.4    1948    98.2 1933.36  150.841912.438
   160.3 1908.57   166.8 1907.45   176.7 1908.09   190.81911.242   199.6 1911.04
     229  1903.6   258.4 1904.72   271.5 1903.68   281.4 1903.01  284.761903.714
   291.2 1906.47   333.7 1905.49   346.8 1906.54   359.9 1906.35   379.5 1909.33
   392.6  1915.4   405.6 1917.49     435 1924.69   451.3 1929.31   467.6 1935.15
   496.9 1946.91   519.7 1957.98   539.3 1965.43   545.8 1969.16   568.6 1979.23
#Mann= 5 ,-1 , 0
       0     .12       0  150.84    .016       0   190.8     .12       0
   271.5    .045       0  284.76     .12       0
#XS Ineff= 2 , 0
                          291.64         1908.11
Permanent Ineff=
       F       F
Bank Sta=271.5,284.76
XS Rating Curve= 0 ,0
Exp/Cntr=0.3,0.1

Type RM Length L Ch R = 1 ,6020    ,340.7,336.2,331.4
XS GIS Cut Line= 4
     2051248.185      270022.427     2051124.921      269897.427
      2051045.06      269755.066      2050857.56      269619.649
#Sta/Elev= 30
       0 1982.72    29.3 1972.09    48.8 1964.04    58.5 1959.02    68.3 1953.07
    81.3  1943.9   126.8 1907.07   133.3 1904.89   146.3 1902.64  175.09 1901.46
   185.4 1899.46   208.2 1900.46  213.371897.288  215.371895.932   221.3 1894.51
   229.81895.916   247.4 1898.66   253.9 1900.42   263.7 1899.59   276.8 1900.82
   286.6 1904.57   296.3  1906.1   322.5 1906.44   345.3  1908.9   384.4 1909.35
     430 1916.59   446.3 1919.48   475.6 1926.24   560.3 1950.03   570.1 1953.51
#Mann= 5 ,-1 , 0
       0     .12       0  175.09    .016       0  213.37     .12       0
  215.37    .045       0   229.8     .12       0
Bank Sta=215.37,229.8
XS Rating Curve= 0 ,0
Exp/Cntr=0.3,0.1

Type RM Length L Ch R = 1 ,5683.7  ,151.6,152.3,152.7
XS GIS Cut Line= 3
     2051406.171      269946.038      2051442.63      269772.427
      2051201.31      269492.913
#Sta/Elev= 30
       0 1978.15      29 1968.97    48.4 1959.86   122.6 1916.21  149.791903.135
   154.8 1900.75   164.5 1893.33   167.7 1891.93  189.131891.987   200.3 1891.18
   223.2 1884.27  228.861883.386   236.2  1882.9   242.8 1883.37   252.6 1887.51
   262.4 1889.66   275.4 1887.88     295 1888.52   314.6 1885.72   327.7 1886.69
   337.5    1885   357.1  1888.8   370.2 1889.24   399.6 1895.27   412.7 1897.18
     429 1897.85   445.4  1897.1     478 1898.95  528.11 1900.15   546.7  1901.8
#Mann= 6 ,-1 , 0
       0     .12       0  149.79    .016       0  189.13     .12       0
  228.86    .045       0   242.8     .12       0  528.11     .06       0
#XS Ineff= 2 , 0
                          260.68         1892.67
Permanent Ineff=
       F       F
Bank Sta=228.86,242.8
XS Rating Curve= 0 ,0
Exp/Cntr=0.3,0.1

Type RM Length L Ch R = 1 ,5531.5  ,133.3,135.6,137.6
XS GIS Cut Line= 3
     2051529.058      269809.172     2051579.855      269712.515
     2051365.657      269451.005
#Sta/Elev= 30
       0 1896.55    12.8 1894.06   24.83 1892.74    57.8 1889.31    80.3 1890.89
    92.11890.718   128.7  1889.9   148.2  1883.4   154.7 1882.12     171 1883.62
   203.4 1884.19   216.4 1880.06   232.7 1879.55   239.2 1878.07   245.7 1877.75
  252.871878.072   255.5 1878.59     262 1882.09   265.2 1882.81   278.2 1883.35
   310.7 1880.66   330.2 1879.79   349.7 1880.31   356.2 1882.61     366 1890.07
   369.2 1891.55   375.7 1892.35   411.5 1892.23  429.231890.974   447.2 1891.37
#Mann= 6 ,-1 , 0
       0     .06       0   24.83    .016       0    92.1     .12       0
   239.2    .045       0  252.87     .12       0  429.23     .06       0
#XS Ineff= 2 , 0
                          278.64         1883.95
Permanent Ineff=
       F       F
Bank Sta=239.2,252.87
XS Rating Curve= 0 ,0
Exp/Cntr=0.3,0.1

Type RM Length L Ch R = 1 ,5395.8  ,220.5,221.8,222
XS GIS Cut Line= 3
     2051697.243      269668.113     2051539.908      269433.738
     2051463.954      269395.761
#Sta/Elev= 30
       0 1883.19    22.7 1884.09    31.9  1883.7    45.4 1884.92    58.4 1884.81
    64.9 1881.73    74.6 1875.15    81.1 1872.99    90.8 1872.96   100.6 1875.38
   116.8 1875.27   139.5 1876.24   152.5 1875.13   161.11873.057   168.7 1872.49
   175.2 1873.06   178.5 1874.66   181.7 1877.02     185 1878.26   188.2 1878.48
   197.9 1877.11   220.6 1875.44   246.6 1875.75   262.8 1879.32   269.3 1880.22
   295.4 1880.56   318.2 1881.68     328  1883.4   344.3 1888.64   367.2 1890.28
#Mann= 4 ,-1 , 0
       0    .016       0    31.9     .12       0   161.1    .045       0
   175.2     .12       0
#XS Ineff= 2 , 0
          142.83 1876.76  186.17         1879.25
Permanent Ineff=
       F       F
Bank Sta=161.1,175.2
XS Rating Curve= 0 ,0
Exp/Cntr=0.3,0.1

Type RM Length L Ch R = 1 ,5174    ,257,261.4,264.7
XS GIS Cut Line= 2
     2051848.068      269584.563     2051686.393       269307.87
#Sta/Elev= 30
       0 1876.45     9.8  1876.4    39.2 1874.22    55.6 1875.43    62.1  1875.3
    65.4 1874.62    68.7 1873.07    75.2 1867.41    78.5 1865.85    81.8 1865.12
    88.3 1864.49   95.21 1865.13   104.6 1866.79   124.3 1866.69   130.8 1866.21
   150.4 1867.99   166.8  1867.5   179.8 1868.88   189.7 1868.57   199.5 1866.39
   202.7 1866.43   209.3 1868.12   219.1 1872.28   222.4 1873.25   225.6 1873.54
   255.1    1873   281.2 1870.56   297.6 1872.19   310.6 1872.04   320.5 1872.53
#Mann= 3 ,-1 , 0
       0     .12       0    81.8    .045       0   95.21     .12       0
#XS Ineff= 2 , 0
                           151.7         1869.58
Permanent Ineff=
       F       F
Bank Sta=81.8,95.21
XS Rating Curve= 0 ,0
Exp/Cntr=0.3,0.1

Type RM Length L Ch R = 1 ,4912.6  ,109.5,112.1,113.7
XS GIS Cut Line= 2
     2052056.401      269503.183     2051950.065      269213.469
#Sta/Elev= 30
       0  1858.7     .551858.815    22.7 1861.29      26 1861.14    35.7 1857.95
    42.2  1856.7    58.5 1858.06    68.2 1855.66    87.7 1856.95   100.7 1855.98
   107.2 1856.12  113.41 1855.29   120.2  1854.7   127.1 1855.25   152.7 1859.21
   162.4 1859.28   175.4 1857.93   181.9 1859.18   188.4 1861.81   194.9  1863.2
   224.2 1861.34   240.4 1861.69   259.9 1861.11   266.4 1862.02   282.6 1868.57
   289.1 1870.27   292.4 1870.73   302.1  1869.8  306.611870.577   308.6 1871.13
#Mann= 5 ,-1 , 0
       0    .016       0     .55     .12       0  113.41    .045       0
   127.1     .12       0  306.61    .016       0
#XS Ineff= 2 , 0
            61.4 1858.86
Permanent Ineff=
       F       F
Bank Sta=113.41,127.1
XS Rating Curve= 0 ,0
Exp/Cntr=0.3,0.1

Type RM Length L Ch R = 1 ,4800.5  ,149.9,152.3,153.7
XS GIS Cut Line= 3
     2052139.044      269481.592      2052070.41      269233.365
     2052012.071      269201.336
#Sta/Elev= 30
       0 1853.88    4.591854.136      13 1853.85    22.8 1852.24    32.6 1852.41
    39.1  1851.9   47.481852.518    58.7 1852.55    78.2 1851.05      88 1852.88
   101.1 1853.15   107.6 1852.89   117.4 1850.51   130.4 1851.21   136.9 1850.99
     150 1853.14   153.2 1853.11   159.7 1851.54   166.3 1850.62   172.8 1850.81
     176 1851.56   185.8 1855.89   195.6 1858.15   205.4 1858.49   228.2 1856.31
   234.7    1857   244.5 1859.78  256.161860.818   298.7 1862.78   324.1 1864.63
#Mann= 6 ,-1 , 0
       0     .12       0    4.59    .016       0   47.48     .12       0
   159.7    .045       0     176     .12       0  256.16    .016       0
#XS Ineff= 2 , 0
           97.88    1854
Permanent Ineff=
       F       F
Bank Sta=159.7,176
XS Rating Curve= 0 ,0
Exp/Cntr=0.3,0.1

Type RM Length L Ch R = 1 ,4648.2  ,260.4,237.6,213.3
XS GIS Cut Line= 3
     2052253.884      269420.717     2052211.566      269200.448
     2052044.466      269192.853
#Sta/Elev= 30
       0  1848.2   14.761848.239    19.5 1847.64    35.8 1846.57    42.3 1847.35
   56.831846.729      65 1846.84    71.3 1845.28      78 1844.74    86.3 1845.25
      91 1846.24    94.3 1846.48   113.8 1846.01   123.5 1845.04     143 1846.32
   152.8 1846.28   159.3 1847.17  170.731851.724   175.5 1853.16   178.8 1853.48
  197.221853.314   204.8 1853.23   225.41853.833   273.5 1856.05   296.4 1857.45
   335.8  1858.8   352.2 1859.68   358.8  1859.6  373.24 1860.59   391.6 1861.43
#Mann= 9 ,-1 , 0
       0     .12       0   14.76    .016       0   56.83     .12       0
    71.3    .045       0    86.3     .12       0  170.73    .016       0
  197.22     .12       0   225.4     .06       0  373.24     .12       0
#XS Ineff= 2 , 0
           43.76 1847.95  110.22         1848.29
Permanent Ineff=
       F       F
Bank Sta=71.3,86.3
XS Rating Curve= 0 ,0
Exp/Cntr=0.3,0.1

Type RM Length L Ch R = 1 ,4410.6  ,90.1,76.1,61.1
XS GIS Cut Line= 3
     2052551.883      269293.712     2052279.314      269184.337
     2052182.091      269024.614
#Sta/Elev= 30
       0 1927.81    39.2 1907.26      62 1894.76    75.1 1887.15   104.4 1869.01
   120.7 1856.62     124 1853.18   127.3 1847.25   130.5 1840.17  132.64 1838.29
   133.8 1837.19   143.6  1836.9   146.8 1837.12   150.6 1838.18   156.6 1839.95
  167.551839.992     173 1839.83   208.8 1840.98   212.1 1841.32   221.9 1843.78
   241.5 1845.11  250.661846.177   280.6 1850.41   303.5 1851.09   388.8 1851.32
   427.81849.731   447.9 1850.36     461 1851.71   470.8 1854.09   480.7 1854.07
#Mann= 6 ,-1 , 0
       0     .12       0  132.64    .045       0   150.6     .12       0
  167.55    .016       0  250.66     .12       0   427.8    .016       0
#XS Ineff= 2 , 0
                          178.53         1844.53
Permanent Ineff=
       F       F
Bank Sta=132.64,150.6
XS Rating Curve= 0 ,0
Exp/Cntr=0.3,0.1

Type RM Length L Ch R = 1 ,4334.5  ,56.9,56.9,57.4
XS GIS Cut Line= 4
     2052616.241      269260.274     2052468.671       269159.58
     2052371.449      269183.885     2052197.838       268980.76
#Sta/Elev= 30
       0 1945.02    45.5 1923.64    87.7 1902.75   113.7 1889.04   139.7 1874.41
   155.9 1863.53   162.4 1857.98   165.7 1854.62   172.2 1846.64   175.4 1844.16
   178.6 1842.28   185.1 1839.95   201.3 1835.61   207.8 1834.08     211 1833.97
   214.2 1834.32   217.6 1835.61   223.9 1839.08   227.1 1839.63  260.131840.108
   275.6 1840.41   298.4 1843.41   324.5 1844.91   357.1 1848.27   417.11848.723
  453.111849.623   461.4 1849.95   487.4 1848.06  502.43 1848.57   546.1 1853.26
#Mann= 7 ,-1 , 0
       0     .12       0   201.3    .045       0   217.6    .016       0
  260.13     .12       0   417.1    .016       0  453.11     .12       0
  502.43     .06       0
Bank Sta=201.3,217.6
XS Rating Curve= 0 ,0
Exp/Cntr=0.3,0.1

Type RM Length L Ch R = 1 ,4277.7  ,61.9,84,105.6
XS GIS Cut Line= 4
      2052630.13      269227.288     2052449.574       269105.76
     2052352.352      269130.066     2052211.727      268965.135
#Sta/Elev= 30
       0 1939.94    45.5 1919.36   126.7 1877.52   139.7 1868.14   149.4 1860.17
   162.4 1846.64   168.9 1841.66   175.4 1837.56   187.6 1834.46   191.7  1834.5
   198.2 1836.64   201.4 1836.97   224.1 1836.71   227.3 1836.16   233.8 1832.68
   240.3  1831.1   246.7  1831.2  250.45 1832.68  252.021833.748   256.4 1836.33
   266.1 1839.27  286.271841.259   340.5  1846.4  373.221847.835  380.261847.677
   421.21849.458   447.3 1849.12  483.081846.448     499 1847.25   534.6 1850.83
#Mann= 10 ,-1 , 0
       0     .12       0   187.6    .016       0   233.8    .045       0
  250.45    .016       0  252.02     .12       0  286.27    .016       0
  373.22     .12       0  380.26    .016       0   421.2     .12       0
  483.08     .06       0
Bank Sta=233.8,250.45
XS Rating Curve= 0 ,0
Exp/Cntr=0.3,0.1

Type RM Length L Ch R = 1 ,4193.7  ,276.2,274.7,272.5
XS GIS Cut Line= 2
     2052643.897      269206.906     2052307.091      268911.767
#Sta/Elev= 30
       0 1937.71    45.8 1916.66   107.9 1885.95   120.9  1878.9   130.8 1872.68
   147.1 1859.43   156.9 1849.38   166.7 1841.47   173.2 1834.87   176.5 1832.68
   179.8 1831.57     183 1831.69  187.691833.379   196.1 1834.16   212.5 1832.88
  224.331833.006   238.6 1829.22   248.4    1828   261.5 1827.42   264.8    1828
   274.6 1833.69   277.8 1833.94   310.5 1832.07   343.2 1831.35   349.8 1833.11
   359.6    1839   366.1 1841.25  384.641841.896   419.2 1842.57   447.8 1841.88
#Mann= 7 ,-1 , 0
       0     .12       0  187.69    .016       0  224.33     .12       0
   248.4    .045       0   264.8     .12       0  384.64    .016       0
   419.2     .12       0
Bank Sta=248.4,264.8
XS Rating Curve= 0 ,0
Exp/Cntr=0.3,0.1

Type RM Length L Ch R = 1 ,3919    ,264.3,263.7,262.6
XS GIS Cut Line= 3
     2052800.147      269087.114     2052716.814      268916.975
      2052468.55       268736.42
#Sta/Elev= 30
       0 1923.21    16.3 1916.43    42.5 1907.44    62.1 1898.16   101.3 1875.59
   107.8 1871.21   124.1 1864.17   130.7 1860.58   137.2  1855.1     147 1848.23
   156.8 1839.18  162.161835.314   176.4 1825.97   179.6 1824.72   189.4 1826.09
  202.141825.422   222.1  1823.2   228.6 1820.26   231.9 1819.56   248.2 1820.32
   290.7 1822.65   303.8 1821.49   326.6 1821.57   372.3 1823.55   395.2 1825.22
     418 1824.52   450.7 1827.02     467 1833.58   470.3 1834.12   496.4 1833.51
#Mann= 5 ,-1 , 0
       0     .12       0  162.16    .016       0  202.14     .12       0
   228.6    .045       0   248.2     .12       0
#XS Ineff= 2 , 0
                          289.47         1826.25
Permanent Ineff=
       F       F
Bank Sta=228.6,248.2
XS Rating Curve= 0 ,0
Exp/Cntr=0.3,0.1

Type RM Length L Ch R = 1 ,3655.3  ,200.8,203.2,204.9
XS GIS Cut Line= 3
     2052949.453      268911.767     2052909.264      268729.858
     2052617.855      268533.295
#Sta/Elev= 30
       0 1874.35    19.6 1861.52      49 1841.06    62.1 1833.73    68.6 1831.48
    71.9 1830.93   90.631829.181     170 1823.14   202.6    1817  245.071816.876
  245.351816.837   251.4 1815.88   264.4 1817.07  283.181817.111   290.4 1812.76
   295.1  1811.5     310 1810.46  315.56 1811.45     323  1813.1     336 1814.05
   342.5 1815.62   355.5  1817.2   358.8 1818.19     362 1820.05   368.6 1825.02
   371.8 1825.72  409.621825.389  467.551825.897  513.211825.843   537.8 1825.76
#Mann= 10 ,-1 , 0
       0     .12       0   90.63     .06       0  245.07     .12       0
  245.35    .016       0  283.18     .12       0   295.1    .045       0
  315.56     .12       0  409.62     .06       0  467.55    .016       0
  513.21     .06       0
Bank Sta=295.1,315.56
XS Rating Curve= 0 ,0
Exp/Cntr=0.3,0.1

Type RM Length L Ch R = 1 ,3452.1  ,94.4,88.2,81.3
XS GIS Cut Line= 2
      2053133.48      268665.239     2052748.064      268351.003
#Sta/Elev= 30
       0  1845.2      36 1836.57    62.2 1831.32    98.2 1825.83     121 1820.87
   134.1 1818.52   147.2 1817.05   163.6 1815.96   173.4 1813.81   183.2  1812.3
   196.3 1812.22  206.341810.854   215.9 1809.95   222.5 1810.59   235.6  1810.1
   238.8 1809.35   245.4 1806.57   258.5 1805.89   264.6 1806.46   287.9 1810.59
  294.711811.063   320.6 1811.97   330.4 1813.99     337 1814.75   356.6 1814.88
   376.2 1816.74  390.931817.181  425.071816.389   431.8 1816.07   497.3 1816.37
#Mann= 7 ,-1 , 0
       0     .06       0  206.34    .016       0   245.4    .045       0
   264.6     .12       0  294.71     .06       0  390.93    .016       0
  425.07     .06       0
Bank Sta=245.4,264.6
XS Rating Curve= 0 ,0
Exp/Cntr=0.3,0.1

Type RM Length L Ch R = 1 ,3363.9  ,47.1,47,47
XS GIS Cut Line= 4
     2053190.772      268613.156     2053013.689      268441.281
     2052921.675      268403.087     2052815.772      268253.781
#Sta/Elev= 30
       0 1847.51    16.2 1843.05    61.7 1833.22   107.2 1827.05   136.4 1822.39
   159.1    1817   168.8 1815.09   194.8 1811.51   221.21810.277   233.8 1807.56
   269.3 1808.18   272.5 1807.85   280.7 1804.51   285.3 1803.52   291.8 1803.36
   298.2 1803.56   301.4  1804.5   336.8 1810.13  347.661811.275   369.3 1811.32
  384.421813.099  391.931814.708   398.7 1816.45     402 1816.57     415 1816.02
   434.7 1814.46   454.3 1814.41   496.8 1813.25   516.4  1813.3   529.5 1812.09
#Mann= 7 ,-1 , 0
       0     .06       0   221.2    .016       0   280.7    .045       0
   301.4     .12       0  347.66    .016       0  384.42     .12       0
  391.93     .06       0
Bank Sta=280.7,301.4
XS Rating Curve= 0 ,0
Exp/Cntr=0.3,0.1

Type RM Length L Ch R = 1 ,3316.9  ,58.2,70.4,82.2
XS GIS Cut Line= 4
     2053225.494      268576.698     2053048.411      268404.823
     2052956.397      268366.628     2052850.494      268217.323
#Sta/Elev= 30
       0 1847.35    16.2 1843.22    48.7 1836.34   103.9  1827.3   142.9  1819.9
   188.3 1809.31   220.8  1807.8  226.441806.776   230.5 1805.73   233.8 1805.76
     237 1806.62   243.5 1807.24  268.81 1807.42  282.471806.767   288.6 1805.32
  297.04 1801.68   304.6 1801.04   315.3 1801.62   317.5 1802.03   327.1 1806.02
  332.181807.269   352.9 1808.57   359.5 1809.86   375.8 1814.29  389.291814.716
     402 1814.68   457.5 1811.55   490.2 1812.24  508.741811.524   529.5 1812.53
#Mann= 9 ,-1 , 0
       0     .06       0  226.44    .016       0  268.81     .06       0
  282.47    .016       0  297.04    .045       0   315.3    .016       0
  332.18     .12       0  389.29     .06       0  508.74     .12       0
Bank Sta=297.04,315.3
XS Rating Curve= 0 ,0
Exp/Cntr=0.3,0.1

Type RM Length L Ch R = 1 ,3246.5  ,434.7,436,436.5
XS GIS Cut Line= 3
     2053248.633      268534.439     2053087.913      268400.453
     2052910.884      268165.507
#Sta/Elev= 30
       0 1844.18    29.4 1837.82    98.1  1825.3     170 1808.84   209.2 1806.63
  217.951806.798   241.9 1806.69     255 1802.03  259.061801.485   268.1 1802.48
   277.9 1802.44   296.3 1799.83   300.8 1799.54   317.1 1799.82   326.9 1801.59
   330.2 1803.17     340 1810.13   343.3 1811.59   349.8 1812.44  365.251811.783
  401.271810.493  426.881809.261  434.491809.202   457.7 1809.48   467.5 1806.52
   470.7 1806.38   477.3 1808.76   487.1 1814.22   496.9 1821.07   503.4  1823.9
#Mann= 9 ,-1 , 0
       0     .06       0  217.95    .016       0  259.06     .12       0
   296.3    .045       0   317.1     .12       0  365.25     .06       0
  401.27     .12       0  426.88     .06       0  434.49     .12       0
#XS Ineff= 2 , 0
          273.68 1804.59
Permanent Ineff=
       F       F
Bank Sta=296.3,317.1
XS Rating Curve= 0 ,0
Exp/Cntr=0.3,0.1

Type RM Length L Ch R = 1 ,2810.5  ,307,303,297.9
XS GIS Cut Line= 3
     2053409.522      268416.975     2053458.133      268193.017
     2053265.425      267915.239
#Sta/Elev= 30
       0 1842.91    81.8 1833.98   114.6 1827.25   137.5 1824.13  180.151810.933
   193.2 1806.82     203 1805.31   216.1 1801.17   235.7 1798.83   258.4 1799.35
   264.9 1798.11  270.261794.949   281.2 1787.17   287.7 1784.53   294.2 1783.18
   320.2 1783.14   349.4 1785.35   365.7 1784.42   378.1 1781.58   388.5 1780.26
     395 1780.55   398.2 1781.62   404.7 1788.54   411.2 1791.42   466.5 1789.74
   479.5 1792.77   495.7 1793.25   521.7 1796.41   547.8 1804.04   567.2 1812.31
#Mann= 5 ,-1 , 0
       0     .06       0  180.15    .016       0  270.26     .12       0
   378.1    .045       0   398.2     .12       0
#XS Ineff= 2 , 0
          347.99 1787.45
Permanent Ineff=
       F       F
Bank Sta=378.1,398.2
XS Rating Curve= 0 ,0
Exp/Cntr=0.3,0.1

Type RM Length L Ch R = 1 ,2507.5  ,300.2,312.6,324
XS GIS Cut Line= 2
     2053807.091      268133.989     2053475.494      267816.281
#Sta/Elev= 30
       0 1793.63    16.4 1791.29    32.8 1785.64    42.6  1785.5    52.5 1783.62
      59  1785.1    72.2 1785.14    88.6 1787.63   111.5 1786.26  132.921783.876
   160.7 1783.59  174.481782.322     187 1782.16   196.8 1776.69   209.9 1771.72
   219.8 1770.82   229.6 1771.74   239.5 1775.54   252.6 1777.74   275.5 1776.47
   291.9 1780.08   314.9 1782.22   360.8 1784.31   377.2 1783.77   387.1 1785.26
   396.9 1782.73   416.6  1782.2     433 1785.23   446.1 1789.33   459.2 1795.98
#Mann= 5 ,-1 , 0
       0     .06       0  132.92    .016       0  174.48     .12       0
   209.9    .045       0   229.6     .12       0
Bank Sta=209.9,229.6
XS Rating Curve= 0 ,0
Exp/Cntr=0.3,0.1

Type RM Length L Ch R = 1 ,2195    ,320.7,312.8,304.6
XS GIS Cut Line= 3
     2053933.828      268010.725      2053843.55      267706.906
     2053748.064      267590.587
#Sta/Elev= 30
       0 1785.09    65.4 1776.17   90.67 1774.36   124.2 1774.31   127.4  1773.9
  134.451770.851   140.5 1768.86   156.8 1770.03   166.6 1771.56   173.2 1774.32
   179.7 1774.99   202.6 1771.96   212.4 1768.92   228.7 1766.25     232 1765.37
   235.3 1763.28   241.8 1762.65   254.9 1763.21   264.7 1763.49   267.9 1764.83
   277.7 1772.32   284.3 1773.73   323.5 1771.24   336.6    1772   346.4 1771.15
   356.2 1773.08   382.4 1781.15   421.6 1795.85   447.8  1807.5   467.4  1818.7
#Mann= 5 ,-1 , 0
       0     .06       0   90.67    .016       0  134.45     .12       0
   235.3    .045       0   254.9     .12       0
Bank Sta=235.3,254.9
XS Rating Curve= 0 ,0
Exp/Cntr=0.3,0.1

Type RM Length L Ch R = 1 ,1882.2  ,315.9,301.9,287.8
XS GIS Cut Line= 2
      2054281.05      267880.517     2053954.661      267449.962
#Sta/Elev= 30
       0 1792.64     4.81791.623   111.3  1778.8   163.7 1773.76  170.141772.032
   176.8  1769.1   186.6 1770.42   199.7 1770.09   209.6 1767.18  217.281761.605
  225.22 1757.08   229.2 1756.68   242.8 1757.05   291.4 1763.46   317.6 1763.89
     334 1762.97   350.4 1764.51   363.5 1762.31   383.1 1763.54   392.9 1762.25
   399.5 1763.24   412.6 1761.38   438.8 1765.93     465 1768.34   471.5 1770.97
   487.9 1780.23   504.3 1793.48   514.1 1797.12   527.2 1808.25   540.3 1817.54
#Mann= 6 ,-1 , 0
       0    .016       0     4.8     .06       0  170.14    .016       0
  217.28     .12       0  225.22    .045       0   242.8     .12       0
Bank Sta=225.22,242.8
XS Rating Curve= 0 ,0
Exp/Cntr=0.3,0.1

Type RM Length L Ch R = 1 ,1580.2  ,313.5,343.5,371.8
XS GIS Cut Line= 4
     2054565.772      267656.559     2054386.953       267486.42
     2054242.855      267441.281     2054123.064      267311.073
#Sta/Elev= 30
       0 1779.23    29.2 1779.25    48.7 1770.12   64.011774.492      78 1772.98
    94.2 1773.19  117.591775.613   133.2 1772.86   152.6 1764.87   185.1 1762.86
  211.991756.438   220.8 1754.97  248.261754.427  266.911755.472   282.2 1756.92
   285.4 1755.87   291.7 1751.05   298.2 1749.93   311.1 1751.02   349.6 1754.55
   375.3 1753.93   420.8 1755.53   443.7 1752.95   453.5 1754.03   476.5 1753.28
   502.7 1755.58     506 1756.65   512.5 1761.22   545.3 1790.43   574.8 1824.37
#Mann= 8 ,-1 , 0
       0     .06       0   64.01     .08       0  117.59     .06       0
  211.99    .016       0  248.26     .08       0  266.91     .06       0
   291.7    .045       0   311.1     .12       0
#XS Ineff= 2 , 0
                          351.08         1758.09
Permanent Ineff=
       F       F
Bank Sta=291.7,311.1
XS Rating Curve= 0 ,0
Exp/Cntr=0.3,0.1

Type RM Length L Ch R = 1 ,1236.8  ,71.6,83.3,97.3
XS GIS Cut Line= 3
     2054662.994        267495.1      2054445.98      267333.642
     2054456.397       267017.67
#Sta/Elev= 30
       0 1764.34    58.7  1758.2    71.7 1758.34    84.7 1760.48   107.5 1757.18
   130.4 1757.37   140.1 1754.63  193.451749.607   205.3 1748.06   224.9  1748.1
   235.51749.357  261.591751.036   316.1 1750.34   319.4 1749.27   325.9 1743.97
   332.4 1740.88   342.2 1739.78  351.13  1740.9   368.3 1744.59   379.61744.712
   394.3 1747.89   410.6 1747.87  436.641756.095   446.5 1757.61   469.3 1758.39
   508.4 1762.78   534.5 1769.05     554 1768.74   573.6  1772.2   586.6 1773.13
#Mann= 8 ,-1 , 0
       0     .06       0  193.45    .016       0   235.5     .06       0
  261.59     .12       0   332.4    .045       0  351.13     .12       0
   379.6     .06       0  436.64     .12       0
Bank Sta=332.4,351.13
XS Rating Curve= 0 ,0
Exp/Cntr=0.3,0.1

Type RM Length L Ch R = 1 ,1153.5  ,55.3,58.5,63.7
XS GIS Cut Line= 4
     2054702.925      267465.587     2054506.744      267305.864
     2054565.772      267186.073     2054485.911      267010.725
#Sta/Elev= 30
       0 1769.65   32.571762.413    55.1 1759.05    87.6  1755.8   110.3 1757.58
  117.92 1757.13   155.7 1755.33   175.71749.935  201.591747.179  204.931747.024
   217.3 1745.84  265.051746.196   282.3 1744.08   292.1 1739.67   298.6 1737.93
   308.4 1737.61   318.1 1737.92  329.491739.871   337.7 1740.94  348.531740.845
     354 1740.63     367 1742.97  381.451743.475   386.5 1744.23   402.8 1749.53
  413.981751.327   487.8 1753.52   517.2 1758.39  532.731762.878   579.2 1769.46
#Mann= 14 ,-1 , 0
       0     .12       0   32.57     .06       0  117.92     .12       0
   175.7     .06       0  201.59     .08       0  204.93    .016       0
  265.05     .06       0   298.6    .045       0   318.1     .06       0
  329.49    .016       0  348.53     .06       0  381.45     .12       0
  413.98     .06       0  532.73     .12       0
Bank Sta=298.6,318.1
XS Rating Curve= 0 ,0
Exp/Cntr=0.3,0.1

Type RM Length L Ch R = 1 ,1095    ,155,130.3,100.6
XS GIS Cut Line= 4
     2054720.286      267446.489     2054550.147      267311.073
     2054609.175      267191.281     2054529.314      267015.934
#Sta/Elev= 30
       0 1770.39    6.691768.865    35.7 1762.08    87.6 1754.49    97.4 1754.46
   110.4  1756.1  130.551756.565   139.6 1756.33   152.5 1754.62  187.551745.745
   214.2 1745.23  220.021744.631     263 1743.02  269.481740.763  289.181738.116
   295.6 1737.17   305.4 1736.47   315.2  1737.2   324.9 1740.19   331.4 1740.97
   373.9 1740.71  384.181741.976   393.4 1744.53  421.851747.619   445.7 1748.71
     498 1752.44   520.8 1755.93   530.6 1760.13   533.9 1760.68   543.7 1759.55
#Mann= 11 ,-1 , 0
       0     .12       0    6.69     .06       0  130.55     .12       0
  187.55     .08       0  220.02    .016       0  269.48     .12       0
  289.18    .016       0   295.6    .045       0   315.2    .016       0
  384.18     .12       0  421.85     .06       0
Bank Sta=295.6,315.2
XS Rating Curve= 0 ,0
Exp/Cntr=0.3,0.1

Type RM Length L Ch R = 1 ,964.7   ,231.6,221.7,211.8
XS GIS Cut Line= 3
      2054789.73      267378.781     2054666.466      267099.267
     2054544.939      267002.045
#Sta/Elev= 30
       0 1772.22    58.5 1760.93    68.2 1758.39      78 1754.61   84.481753.991
  115.861744.814   146.2  1741.8   178.61740.997   185.2 1739.76     195 1736.31
     208 1736.42   213.5 1735.54   224.2  1733.3     234 1733.47  237.92 1735.54
   240.5 1736.91   243.7  1737.5   253.5 1737.04  276.13 1738.24   308.7 1738.74
  321.771740.966   334.7 1744.29   347.6 1745.98   386.5 1746.65   435.2 1751.65
   441.7 1753.92   444.9 1756.53   448.2 1758.06   454.6 1759.06   461.1 1759.09
#Mann= 8 ,-1 , 0
       0     .06       0   84.48    .016       0  115.86     .06       0
   178.6     .12       0   213.5    .045       0  237.92     .12       0
  276.13    .016       0  321.77     .06       0
#XS Ineff= 2 , 0
                          244.07         1738.61
Permanent Ineff=
       F       F
Bank Sta=213.5,237.92
XS Rating Curve= 0 ,0
Exp/Cntr=0.3,0.1

Type RM Length L Ch R = 1 ,743     ,224.7,219.4,214
XS GIS Cut Line= 2
     2054961.605        267120.1     2054697.716      266887.462
#Sta/Elev= 30
       0  1754.6    22.8 1745.46    42.4 1738.71    48.9  1738.1    55.4 1736.77
    68.4 1736.14  107.84 1736.05   140.1 1735.66   143.3 1735.17   149.8 1733.16
  154.511732.726   159.6 1732.47  163.18 1731.84   166.1 1730.86   172.6 1730.43
   182.4 1730.61   188.9 1731.84   198.7 1732.52   202.31732.439  206.021732.637
   218.2 1732.79   234.5 1734.19   247.6 1734.22  263.051735.165   286.6 1736.57
   293.2 1736.65   309.4 1737.56   332.2 1740.12   345.3 1742.52   351.8 1743.43
#Mann= 8 ,-1 , 0
       0     .12       0  107.84     .06       0  154.51     .12       0
  163.18    .045       0   188.9     .12       0   202.3     .06       0
  206.02    .016       0  263.05     .06       0
#XS Ineff= 2 , 0
                          208.88         1734.48
Permanent Ineff=
       F       F
Bank Sta=163.18,188.9
XS Rating Curve= 0 ,0
Exp/Cntr=0.3,0.1
